HEC-RAS study BeaverCreek.prj: BeaverCreek

--- BeaverCreek.g01 (geometry) --- (continued)

Type RM Length L Ch R = 1 ,9875.521,89.25,91.44,95.12
XS GIS Cut Line= 6
     637970.7219    4336978.9865     637733.6805    4337030.4225
     637600.4022    4337097.9527     637589.3874    4337103.8373
      637582.316    4337108.9603     637264.2829    4337148.8494
#Sta/Elev= 30
       0  963.11   12.28  962.19   15.35  961.63   33.77  959.84   39.91  958.96
   58.34  957.68  101.32  955.28  178.08  952.51  181.15  952.14  184.22  950.92
  187.29  950.43  245.61   949.7  352.33  947.77  385.87  946.51  397.42  945.75
   401.8  945.55  406.82  945.75  419.29  946.52  440.66  947.33  462.03  947.59
  495.61  947.27  523.08  949.36  538.35  950.04  571.93  952.35  587.19  952.71
   599.4     952  614.66  953.75  684.87  957.66  724.56  961.12  733.71   962.3
#Mann= 3 , 0 , 0
       0     .09       0  397.42     .04       0  406.82     .09       0
Bank Sta=397.42,406.82
XS Rating Curve= 0 ,0
Exp/Cntr=0.3,0.1

Type RM Length L Ch R = 1 ,9784.08 ,69.14,91.44,108.77
XS GIS Cut Line= 5
     637967.5469    4336947.2365     637595.2674     4337004.174
     637549.4939    4337021.3708     637544.8768    4337020.9641
     637242.0579    4337105.9868
#Sta/Elev= 30
       0  962.87   21.43  960.67   27.56  959.66   33.68  959.02   70.42  956.33
   94.92  954.91  143.91  953.94  146.97  953.77  159.22  952.19  186.77  950.75
  195.96  949.65  208.21  950.13  272.51   948.5  358.24  947.69  416.34   945.9
  422.45  945.47  425.51  945.71  426.94  946.14  433.19  946.84  445.41  947.32
  488.16  947.74  533.97  949.58  579.77  951.95   604.2  952.25  619.47  952.78
  668.33  956.14  701.92  957.42  726.35  960.22  735.51  961.52  744.67  964.34
#Mann= 3 , 0 , 0
       0     .09       0  416.34     .04       0  426.94     .09       0
Bank Sta=416.34,426.94
XS Rating Curve= 0 ,0
Exp/Cntr=0.3,0.1

Type RM Length L Ch R = 1 ,9692.64 ,97.49,91.44,83.77
XS GIS Cut Line= 6
     637978.6594    4336931.3614     637582.7655    4336960.0781
     637548.7342    4336934.8896     637522.9825    4336925.8903
     637514.0528    4336918.2835     637229.3579    4337025.0241
#Sta/Elev= 30
       0  962.96   12.21  962.37    45.8   958.7   79.39  956.13  119.08  953.91
  155.72  952.63  195.41   950.7  213.73  949.11  219.84  950.05  222.89   950.1
  262.59  948.63  308.39  947.76  338.92  947.49  387.77  947.85  420.62  946.66
   429.5   945.8  435.03  945.24  439.89  945.89  445.85  947.32  448.82   947.5
  459.49  947.05  481.98  946.97  540.33   947.5  571.04  948.29  623.25  950.18
  675.46   953.1  715.39  954.49  752.24  956.97  761.45   957.9  782.95  962.08
#Mann= 3 , 0 , 0
       0     .09       0   429.5     .04       0  439.89     .09       0
Bank Sta=429.5,439.89
XS Rating Curve= 0 ,0
Exp/Cntr=0.3,0.1

Type RM Length L Ch R = 1 ,9601.2  ,63.84,91.44,61.22
XS GIS Cut Line= 5
     638042.1595    4336847.2238     637657.9136    4336875.2213
     637541.3216    4336837.6111     637525.9591    4336851.9501
     637232.5329    4337013.9116
#Sta/Elev= 30
       0  962.87   12.23  962.17   30.58  962.17   48.92  961.07   64.21  960.85
   91.73  959.26  110.08  958.93  192.63  953.15  214.04  952.06  229.32  951.84
  241.55  950.12   259.9  948.65  287.42  947.95  296.59  948.83  305.77   948.9
  333.28  947.64  400.58  946.59  452.64  947.09  458.77   945.5  461.83  944.88
  464.89  944.79  467.96  945.14  477.15  946.67  580.58   947.7  635.43   947.7
  668.94  948.68  815.19  956.57  839.57  958.33  848.71  960.46  863.94  962.36
#Mann= 3 , 0 , 0
       0     .09       0  458.77     .04       0  467.96     .09       0
Bank Sta=458.77,467.96
XS Rating Curve= 0 ,0
Exp/Cntr=0.3,0.1

Type RM Length L Ch R = 1 ,9509.76 ,76.98,91.44,17.81
XS GIS Cut Line= 6
     637975.4844    4336761.4986     637592.2638    4336803.4431
     637562.3658    4336778.5722     637526.3824    4336791.8014
     637510.5074    4336788.3618     637234.1204    4337001.2116
#Sta/Elev= 30
       0  963.19   27.54  961.55   73.43  957.61  116.26   954.7  171.34  952.08
  217.23  949.27  253.95   948.7  275.36  946.88  357.97  946.56  406.15  944.86
  410.86  944.74  413.21  944.94  419.03  945.61   439.6  945.42  460.24  946.22
  479.44  946.16  522.28  947.04     559  948.38  623.26     949  641.62  950.14
  659.98  950.66  721.18  953.39  733.42  954.32  748.72  955.95   773.2  956.88
  794.63  958.67  806.87  959.33  812.99  960.08  822.17  962.14  828.29   962.8
#Mann= 3 , 0 , 0
       0     .09       0  406.15     .04       0  413.21     .09       0
Bank Sta=406.15,413.21
XS Rating Curve= 0 ,0
Exp/Cntr=0.3,0.1

Type RM Length L Ch R = 1 ,9418.32 ,139.64,91.44,3.67
XS GIS Cut Line= 6
     638002.1346    4336684.6039     637598.1243    4336737.7654
     637570.6076    4336704.6925      637551.293    4336711.8362
     637514.4136    4336779.9724      637224.258    4336995.7545
#Sta/Elev= 30
       0  965.04   49.02  961.61   79.66  960.29   91.92     959  104.17  958.79
  125.62  957.68  147.07  955.71  165.45  955.08  281.87  948.91  294.13  948.62
  318.64  947.03  346.22  946.27  370.73  946.81  442.75  944.63  452.46  944.68
     479  945.24  502.75  944.55  523.54  944.74  548.56  945.88  596.64  946.89
  639.54   948.4  703.89   949.2  716.15  950.17  762.12   951.7  808.08  954.04
  829.53  956.41  850.98   956.8  866.31  957.93  893.89  960.43  912.27  963.41
#Mann= 3 , 0 , 0
       0     .09       0  442.75     .04       0  452.46     .09       0
Bank Sta=442.75,452.46
XS Rating Curve= 0 ,0
Exp/Cntr=0.3,0.1

Type RM Length L Ch R = 1 ,9326.88 ,3.36,91.44,79.26
XS GIS Cut Line= 6
     637838.6218    4336390.9158     637517.6776    4336656.3133
     637522.8034    4336683.5242     637546.4745    4336710.6757
     637510.6926    4336779.7152      637221.083     4336984.642
#Sta/Elev= 30
       0  962.85   12.25  961.67    88.8  957.79  128.61  954.33  192.92  952.14
  235.79  949.79  248.04  949.86  263.35   948.1  278.66  947.67   300.1  946.36
  315.41  947.23  379.72  945.72  416.46  945.67  462.16  944.86  471.17  944.82
   486.1  945.17  509.79  944.46  527.55  944.64  553.52  945.79  607.01     947
  652.89  948.59  704.88  949.25  723.23  950.39  756.88  951.33  811.93  954.14
  836.39  956.07   857.8  956.38   873.1  958.47  897.56  960.19  912.86  962.59
#Mann= 3 , 0 , 0
       0     .09       0  462.16     .04       0  471.17     .09       0
Bank Sta=462.16,471.17
XS Rating Curve= 0 ,0
Exp/Cntr=0.3,0.1

Type RM Length L Ch R = 1 ,9235.44 ,95.72,91.44,8.14
XS GIS Cut Line= 6
     637829.0967    4336382.9783     637514.1851    4336652.9266
     637520.1264    4336695.1643     637451.3464    4336731.9711
     637432.8256    4336754.4607     637206.7955     4336975.117
#Sta/Elev= 30
       0  962.84   30.72  960.62   92.17  957.43   122.9  955.03   144.4   953.7
   178.2  952.78  227.36  950.32  245.79  949.83   267.3  947.89  291.88  947.02
  298.03  946.52   301.1  946.57  307.24  947.26  313.39  947.28  384.05  945.67
  423.92  945.69  454.39  944.96  490.67  944.79  502.76  944.47  505.78  944.37
  511.82  944.56   538.4  945.04  555.88  946.91  567.69  947.66  647.42  949.43
  705.69   951.1  767.02  953.78  834.49  957.89  868.23  961.68  880.49   964.2
#Mann= 3 , 0 , 0
       0     .09       0  502.76     .04       0  511.82     .09       0
Bank Sta=502.76,511.82
XS Rating Curve= 0 ,0
Exp/Cntr=0.3,0.1

Type RM Length L Ch R = 1 ,9144    ,23.44,91.44,110.3
XS GIS Cut Line= 6
     637754.4841    4336330.5907     637438.5042    4336614.3569
     637422.4656    4336695.4455        637447.5    4336718.3384
     637427.9208    4336749.2947     637197.2705     4336962.417
#Sta/Elev= 30
       0  963.25   21.39  961.04   45.83  959.07      55   957.9   76.38  956.16
  122.21  953.37  140.55  953.57  149.71  953.35  174.16   952.3  204.71  950.17
  223.04  950.73  278.04   947.9  293.32  948.05  329.98  946.62  357.48  945.93
   369.7  945.21  429.99  945.43  471.25  944.29  495.48  944.58  515.95   944.4
  524.29  944.35  564.64  944.79   573.8  945.32  586.01  946.63  601.27  947.76
  680.54  949.52   796.4  953.47  848.23  956.79  897.01  961.33  909.21  962.73
#Mann= 3 , 0 , 0
       0     .09       0  515.95     .04       0  524.29     .09       0
Bank Sta=515.95,524.29
XS Rating Curve= 0 ,0
Exp/Cntr=0.3,0.1

Type RM Length L Ch R = 1 ,9052.561,52.68,91.44,100.09
XS GIS Cut Line= 6
     637748.1341    4336313.1282     637436.2161    4336605.8728
     637419.4145    4336610.9482     637411.5329    4336644.8435
     637329.5387    4336673.3632     637133.7703    4336898.9168
#Sta/Elev= 30
       0  963.26   12.22  962.05   36.67  960.69   91.67  955.77  106.94  955.47
  122.22   953.9  143.61  953.73  161.94  953.03  210.83  949.87  216.94  949.92
  223.05  950.77  232.22  950.93  259.72   948.7  293.33  947.74  305.55  948.07
  378.89  945.08   430.7  945.37   492.1  944.34  495.09   944.3  501.08  944.41
  519.04  945.95  531.02  946.48  588.27  948.53  609.61  948.68  652.27  949.92
  688.84  951.67   807.7  955.99  835.13  957.93  856.46  961.63   865.6  962.48
#Mann= 3 , 0 , 0
       0     .09       0   492.1     .04       0  501.08     .09       0
Bank Sta=492.1,501.08
XS Rating Curve= 0 ,0
Exp/Cntr=0.3,0.1

Type RM Length L Ch R = 1 ,8961.12 ,116.64,91.44,42.81
XS GIS Cut Line= 6
     637654.4714    4336319.4782     637422.7668    4336553.0837
     637396.8904    4336565.9425     637355.5526    4336560.2058
     637318.6265    4336570.2287     637125.8328    4336894.1543
#Sta/Elev= 30
       0  963.02   24.37  960.02   51.79  957.95   79.21  955.11    91.4  954.67
  109.68  952.53     131  951.91  149.28  949.52  164.51  950.91  204.12  947.73
  213.26  947.88  237.63     947  249.82  947.37  277.24  945.75  325.98  944.67
  374.39  944.29  385.56  944.29  515.32  946.62  533.71  947.79  555.17  948.08
  591.94  949.45  625.65  951.59  671.62  953.26  686.95   954.5  699.21  954.07
  745.18  955.38  766.63  957.07  775.82  958.71  794.21  961.01  815.67  962.98
#Mann= 3 , 0 , 0
       0     .09       0  374.39     .04       0  385.56     .09       0
Bank Sta=374.39,385.56
XS Rating Curve= 0 ,0
Exp/Cntr=0.3,0.1

Type RM Length L Ch R = 1 ,8869.68 ,106.61,91.44,33.89
XS GIS Cut Line= 5
     637417.9334    4336267.0906     637335.3212    4336478.5889
      637307.085    4336535.0618     637297.7509    4336548.9156
     637125.8328    4336879.8668
#Sta/Elev= 30
       0  963.36   33.75   960.9   42.96  959.71   52.16     958  110.46  952.18
   125.8  951.43  147.28  948.96  168.76  947.92  199.44  947.48  236.08  944.53
  239.09  944.26   245.1  944.55  272.16  945.42  287.19  945.22  316.07   945.8
  352.76  945.65   371.1  946.46  410.84  947.51  444.46  949.07  453.63   948.9
  468.92  949.92  490.32  950.66  517.83  952.52   548.4  952.95  578.97  954.62
  603.42  954.69  618.71  955.65  627.88  957.21  649.27  959.61  679.84  962.41
#Mann= 3 , 0 , 0
       0     .09       0  236.08     .04       0   245.1     .09       0
Bank Sta=236.08,245.1
XS Rating Curve= 0 ,0
Exp/Cntr=0.3,0.1

Type RM Length L Ch R = 1 ,8778.24 ,69.94,91.44,108.38
XS GIS Cut Line= 6
     637225.8455    4336228.9905     637227.5303    4336460.4529
     637242.4754    4336495.2039     637262.1908    4336521.0426
     637279.3888    4336554.6447     637119.4828    4336865.5793
#Sta/Elev= 30
       0  964.05    3.05  962.06    6.09  960.79   12.18  959.72   21.32  957.55
   51.78   954.4      67  953.66   85.28  952.04   94.41  951.54  124.87  951.68
  170.56  948.36  188.83  948.14  231.47  945.93  260.57  944.67  278.32  944.23
  282.92  944.23  293.16  944.23  339.63  945.56  382.57  945.61  394.84  946.42
  462.31  948.58  477.65  948.82  489.92   949.8  545.12  952.51  572.73  952.99
   603.4  955.58  637.13  957.54  643.27  958.29   649.4  959.62  689.27  962.79
#Mann= 3 , 0 , 0
       0     .09       0  282.92     .04       0  293.16     .09       0
Bank Sta=282.92,293.16
XS Rating Curve= 0 ,0
Exp/Cntr=0.3,0.1

Type RM Length L Ch R = 1 ,8686.8  ,37.99,91.44,113.76
XS GIS Cut Line= 6
     637213.1455    4336225.8155     637165.9109    4336526.6112
     637171.1032    4336548.4904     637171.6957    4336552.7173
     637171.8641    4336589.7145     637068.6827    4336857.6417
#Sta/Elev= 30
       0  962.23   15.22  959.67    27.4  958.36   39.58  957.67   45.67  956.96
   54.81  955.29    60.9  954.63   70.03   954.2   91.34  952.43  106.57  951.55
  127.88  951.25  152.24  949.14  167.46  948.17   176.6  948.37  188.78  947.98
  246.63  945.52  277.08  944.84  325.13  944.31   329.1  944.23  334.08  944.28
  404.89  947.17  444.59  949.23  478.19  951.26  508.73  953.53  527.06  955.45
  539.28  956.23   591.2  959.18  606.47  960.29  637.02  961.04  655.34  962.48
#Mann= 3 , 0 , 0
       0     .09       0  325.13     .04       0  334.08     .09       0
Bank Sta=325.13,334.08
XS Rating Curve= 0 ,0
Exp/Cntr=0.3,0.1

Type RM Length L Ch R = 1 ,8595.36 ,137.96,91.44,47.53
XS GIS Cut Line= 6
     637155.4662    4336230.8955     637144.0497    4336483.8478
     637111.2081    4336504.8496     637088.1668    4336511.1168
     637065.4683    4336538.6167     637002.0076    4336846.5292
#Sta/Elev= 30
       0  962.99     6.1  963.07    9.15  962.48   24.41  957.52   33.56  956.18
   36.61  956.13   48.81  954.71   61.01   953.9   91.52  952.18  112.88  951.41
  122.03  950.38  128.13  950.05  149.49  948.15  155.59   947.9  167.79  948.18
  241.01   945.4  295.18  944.25  298.16  944.23  304.13  944.23  397.51  946.21
  421.93  947.97  470.77  950.13  492.13  951.56   513.5   953.4  534.86  954.31
  547.07  955.18  586.75  956.86  611.17  959.14   647.8   961.3  666.11  962.88
#Mann= 3 , 0 , 0
       0     .09       0  295.18     .04       0  304.13     .09       0
Bank Sta=295.18,304.13
XS Rating Curve= 0 ,0
Exp/Cntr=0.3,0.1

Type RM Length L Ch R = 1 ,8503.92 ,82.65,91.44,64.16
XS GIS Cut Line= 6
      637022.116    4336136.7036     637009.9306    4336479.0329
     637015.8527    4336496.3202     637015.6472    4336501.2575
     637025.7609    4336544.6161      636979.077    4336840.1439
#Sta/Elev= 30
       0  961.81    6.12  962.39   18.35  961.84   51.99  957.47   58.11  956.92
   76.46  957.04  100.93  956.34  134.57  956.08  143.75  955.38  149.86  954.13
  152.92  953.45  155.98  951.88  159.04  950.84  180.45  950.84  256.91  947.19
  354.73  944.23  362.36  944.23  425.55  944.77  443.87  946.47  477.45  948.63
  517.14  950.07  575.14  953.72   578.2  953.72  596.52   955.1  617.89  955.84
  642.31  957.66  663.68  959.75     682   960.5  694.21  961.77  709.48  962.74
#Mann= 3 , 0 , 0
       0     .09       0  354.73     .04       0  362.36     .09       0
Bank Sta=354.73,362.36
XS Rating Curve= 0 ,0
Exp/Cntr=0.3,0.1

Type RM Length L Ch R = 1 ,8412.48 ,49.88,91.44,133.01
XS GIS Cut Line= 6
     637018.0237    4336127.4608     636928.2805    4336471.7343
     636936.4826     4336486.551     636931.3967    4336530.3001
      636971.143    4336562.7512     636939.7069    4336851.3623
#Sta/Elev= 30
       0   961.8    6.13   960.4     9.2  960.08   21.47  960.21    36.8  958.62
   52.14  958.07   67.48  956.59   92.01   956.9  150.29  955.53  156.42  954.86
  165.62  950.87  184.02  950.58   233.1  947.58  254.57  947.09   279.1  947.45
  355.78  945.14  405.01  944.23  421.87  944.23  433.54  944.23  459.57  945.27
  468.61  945.28  526.68  948.97  603.08  952.04  624.47  953.72  639.75  955.99
  655.03  955.54  679.48  957.52  725.32   960.4  746.71  962.06  758.93  963.37
#Mann= 3 , 0 , 0
       0     .09       0  421.87     .04       0  433.54     .09       0
Bank Sta=421.87,433.54
XS Rating Curve= 0 ,0
Exp/Cntr=0.3,0.1

Type RM Length L Ch R = 1 ,8321.04 ,31.89,91.44,95.18
XS GIS Cut Line= 6
     637007.4404    4336118.9942     636892.5705    4336462.1586
     636873.0492    4336505.3722     636849.3904     4336531.797
      636833.784    4336552.8358     636802.1233    4336868.2957
#Sta/Elev= 30
       0  963.17   12.27  960.64   21.47  957.45   24.53  957.32   30.67  958.44
   33.73  958.49   42.93  957.07   70.54  956.12   101.2  956.79   110.4  956.53
  113.47   955.9   119.6  955.84   128.8  954.76  150.27  954.35  159.47  952.88
  168.67  950.22  190.14  950.34  202.41  949.21  245.34  947.02  294.41  947.18
  373.73  944.56  400.41  944.23  433.01  944.23  442.37  944.23  483.26  946.35
  626.54  951.32  690.56  954.33  748.48  957.88  772.87  961.46  788.11  963.07
#Mann= 3 , 0 , 0
       0     .09       0  433.01     .04       0  442.37     .09       0
Bank Sta=433.01,442.37
XS Rating Curve= 0 ,0
Exp/Cntr=0.3,0.1

Type RM Length L Ch R = 1 ,8229.601,140.13,91.44,18.84
XS GIS Cut Line= 6
     636998.9737    4336083.0107     636872.5415     4336454.565
     636805.6713    4336478.6923     636788.0069    4336452.9775
     636754.2725    4336503.3807     636736.5065     4336897.929
#Sta/Elev= 30
       0  962.43    6.13  960.93    18.4  959.64   30.66  960.73   36.79  960.63
   55.19  956.22   70.52  955.87   85.85  953.15  110.38  952.03  125.72  949.99
  211.57  950.15   226.9  948.35   245.3  947.56  288.22   946.8  334.22   946.9
  410.25  944.23  471.72  944.23  485.27  944.23  562.64  945.19  734.09   949.6
  758.58  949.66  813.69  952.71  832.06  952.82  856.55  954.36  874.92  954.55
  890.23  956.92  893.29  956.94  917.79  961.27  933.09  962.45  951.46  963.02
#Mann= 3 , 0 , 0
       0     .09       0  471.72     .04       0  485.27     .09       0
Bank Sta=471.72,485.27
XS Rating Curve= 0 ,0
Exp/Cntr=0.3,0.1

Type RM Length L Ch R = 1 ,8138.16 ,63.39,91.44,64.58
XS GIS Cut Line= 6
     636998.9737     4336061.844       636835.99    4336218.4777
      636757.518    4336395.2806     636778.6704    4336454.4154
     636745.0826    4336489.4725     636723.8065    4336912.7457
#Sta/Elev= 30
       0  964.55   15.27  958.75   24.44  957.37   54.98  955.39   76.37  958.27
   82.48  959.86   88.59   960.1  134.41  954.37  152.74  950.87  180.23  948.09
  213.83  948.78  229.12  947.83  247.54  950.06  259.82  947.67  281.32  947.91
  296.67  946.22  358.08  945.32  422.48  945.69  470.56  944.23  477.27  944.23
   519.1   944.5  654.07  947.34  755.42  950.77  773.85   950.5  801.48  951.81
  816.84  951.83  838.34  954.08  865.98  954.46  908.97  961.14  955.04  962.95
#Mann= 3 , 0 , 0
       0     .09       0  470.56     .04       0  477.27     .09       0
Bank Sta=470.56,477.27
XS Rating Curve= 0 ,0
Exp/Cntr=0.3,0.1

Type RM Length L Ch R = 1 ,8046.72 ,103.67,91.44,64.95
XS GIS Cut Line= 6
     636994.7403    4336051.2607     636812.7066     4336210.011
     636700.2489    4336404.2235     636681.4823    4336471.1738
     636670.3678    4336679.8842      636668.773    4336974.1292
#Sta/Elev= 30
       0  962.96    6.11  960.42   18.34  958.98   45.86  957.27   55.03  957.75
   67.26  959.81   82.55  960.16  110.07  956.27   143.7  950.08  149.81  949.41
  177.33  949.82  204.84  949.32  220.13  950.01  241.53   948.5   256.7  950.25
  265.79  949.85  274.89  948.44  290.06  948.75  326.45  946.35  420.46  945.91
  516.14  944.25  517.42  944.14  523.19  944.28  709.76  947.54  737.42  948.43
  795.68  950.58  866.18  954.11  942.81  959.54 1019.43  961.63 1040.89  963.08
#Mann= 3 , 0 , 0
       0     .09       0  516.14     .04       0  523.19     .09       0
Bank Sta=516.14,523.19
XS Rating Curve= 0 ,0
Exp/Cntr=0.3,0.1

Type RM Length L Ch R = 1 ,7955.28 ,73.92,91.44,70.86
XS GIS Cut Line= 6
     637011.6737    4336019.5106     636601.4268     4336364.095
     636601.3729    4336406.5075     636611.4221    4336480.5916
     636622.0643    4336512.2619      636656.073    4336986.8292
#Sta/Elev= 30
       0  963.08   36.74  960.54   64.29  959.68   88.78  961.37  107.15  961.63
  113.28  961.13  165.32   950.6  168.38  950.35  241.86  951.52  260.23  950.55
   278.6  948.64  284.72  948.65  300.03  950.46  306.15  950.18   318.4  948.32
  434.73  946.32  547.88  945.73     560  945.22  569.09  945.48  605.09  943.93
  608.08  943.85  614.06  943.96  827.55  947.15  910.43  950.18  968.75  953.04
 1011.72  956.54 1027.07  956.82 1048.56  958.79 1137.58  961.57 1162.14  963.06
#Mann= 3 , 0 , 0
       0     .09       0  605.09     .04       0  614.06     .09       0
Bank Sta=605.09,614.06
XS Rating Curve= 0 ,0
Exp/Cntr=0.3,0.1

Type RM Length L Ch R = 1 ,7863.84 ,102.13,91.44,58.85
XS GIS Cut Line= 6
     636994.7403     4336017.394     636527.5021    4336385.7909
     636527.2904    4336439.5543     636512.5004    4336448.3312
     636570.9044    4336562.0064     636645.4896    4336997.4126
#Sta/Elev= 30
       0   962.5   21.47  962.35   46.01  960.72   67.47  962.36   76.68  963.55
   85.88  963.69  107.35  960.16  138.02  953.59  144.15  951.34  147.22  951.17
  171.75  952.69  214.69  952.82  233.09  953.36   251.5  952.33   279.1  948.66
   297.5   950.6  303.64   950.4   315.9  948.56  358.84  947.35  456.99  946.13
  582.73  945.86  648.77  943.74  652.18  943.74  661.33  943.74  705.87  943.79
  889.21  946.89  987.37  950.72 1103.95  957.91 1159.16   959.1 1235.86  962.95
#Mann= 3 , 0 , 0
       0     .09       0  652.18     .04       0  661.33     .09       0
Bank Sta=652.18,661.33
XS Rating Curve= 0 ,0
Exp/Cntr=0.3,0.1

Type RM Length L Ch R = 1 ,7772.4  ,82.21,91.44,66.11
XS GIS Cut Line= 5
     636969.3403    4336025.8606     636424.1265    4336376.6654
     636428.1902    4336436.1384     636523.1289    4336590.6235
     636607.3896    4337037.6293
#Sta/Elev= 30
       0  962.97   18.44  961.65   39.94  963.28   49.16   964.5   55.31   964.4
   82.96   959.8  110.61  952.23  113.69  951.85  129.05  952.26  159.78  954.41
  212.01  954.46  242.74  953.07  270.39  949.52  276.54  949.41  282.68  950.57
  294.97  950.95  307.26  948.63  316.48  948.38  439.38  947.46  485.47  946.43
  654.28  945.48  732.52  943.74  741.74  943.75  870.82   944.9  935.36  946.03
 1085.96  951.92 1132.07  955.22 1245.79  957.66 1337.99  961.14 1344.14   961.8
#Mann= 3 , 0 , 0
       0     .09       0  732.52     .04       0  741.74     .09       0
Bank Sta=732.52,741.74
XS Rating Curve= 0 ,0
Exp/Cntr=0.3,0.1

Type RM Length L Ch R = 1 ,7680.96 ,12.52,91.44,203.16
XS GIS Cut Line= 6
      636965.107    4336015.2773     636349.8472    4336419.9663
     636359.3912    4336489.3713     636392.9414    4336502.5406
     636452.2412    4336601.7354     636554.4728    4337071.4961
#Sta/Elev= 30
       0  963.24   18.43  961.93      43   964.6   52.21  964.34   79.85  961.05
   92.14  956.38  113.64  952.25  132.06  952.38  147.42  954.46  175.06  956.07
  248.77  953.41  282.56  950.43  300.98  951.24  316.34   948.8  325.55  948.59
  420.76  949.41  485.26  946.67  693.64  945.15  767.87  945.52  812.86  943.76
  816.48  943.74  819.33  943.74  849.59  944.84   864.8  943.75  910.42  944.02
 1029.51  946.18 1234.67  953.63 1344.91   955.4 1390.84  957.19 1439.84  961.25
#Mann= 3 , 0 , 0
       0     .09       0  812.86     .04       0  819.33     .09       0
Bank Sta=812.86,819.33
XS Rating Curve= 0 ,0
Exp/Cntr=0.3,0.1

Type RM Length L Ch R = 1 ,7589.52 ,73.99,91.44,72.03
XS GIS Cut Line= 6
     636960.8736    4336000.4606     636383.1313    4336379.3787
     636337.8875    4336424.2256     636331.1607    4336571.1278
      636281.928    4336599.2479     636186.1721    4336946.6125
#Sta/Elev= 30
       0  963.37    21.5  961.97   39.92  963.87    52.2  963.67  104.41  956.17
  113.62  952.55  116.69  952.35  132.04  952.21  162.75  956.48  184.24  957.05
  236.45  954.93  294.79  950.95  313.22  951.41  334.71  948.74  426.83  950.05
  460.61  949.08  482.11  947.14  700.02  945.05  784.18  945.38  834.52  943.74
  880.34  943.74  886.51  943.74 1088.23  946.07 1118.77  947.81 1164.57  947.54
 1256.17  951.19 1265.34  951.92 1283.66  959.35 1289.76  960.75  1320.3  962.84
#Mann= 3 , 0 , 0
       0     .09       0  880.34     .04       0  886.51     .09       0
Bank Sta=880.34,886.51
XS Rating Curve= 0 ,0
Exp/Cntr=0.3,0.1

Type RM Length L Ch R = 1 ,7498.08 ,9.48,91.44,59.41
XS GIS Cut Line= 6
     636950.9782    4335992.7877     636371.1556     4336370.762
      636347.343    4336371.5558     636273.1509    4336487.0585
     636253.9449    4336530.9014     636096.3194    4336758.7579
#Sta/Elev= 30
       0   962.9    24.5  961.69   39.81  962.39   58.19  961.42   91.88  956.78
  107.19  952.76  119.44  952.25  125.57  952.41     147  956.56  165.38  957.78
  183.75  957.82  232.76  955.59  294.01  951.33  318.51  951.43  330.76  949.71
  339.95  949.49  416.51  950.51  456.32  949.57  468.57  948.31  514.51  948.89
   572.7  946.03  824.81  943.74  849.59  943.74  859.83  943.74   936.9  945.14
 1031.63  950.21 1080.53  951.39 1126.36  954.72 1163.04  956.11 1178.31  961.13
#Mann= 3 , 0 , 0
       0     .09       0  849.59     .04       0  859.83     .09       0
Bank Sta=849.59,859.83
XS Rating Curve= 0 ,0
Exp/Cntr=0.3,0.1

Type RM Length L Ch R = 1 ,7406.64 ,3.49,91.44,110.04
XS GIS Cut Line= 6
     636944.3636    4335986.1731     636348.2073    4336361.9646
     636285.8978     4336424.671     636176.6899    4336471.4398
     636190.2508    4336540.1619     636076.8435     4336744.628
#Sta/Elev= 30
       0  962.78    55.3  960.38   79.88  957.92  101.39  953.28  116.75  952.31
  122.89  952.63  141.33  956.74  159.76  957.71  187.41     958  294.95  951.65
   322.6  951.44  337.96   949.9  411.69   950.9  454.71  949.53  463.92  948.49
  506.94  949.54  537.66  948.83  571.46  946.25  778.27  943.74  923.07  943.74
  931.01  943.74  981.28  944.13 1026.62  947.17 1044.84   949.4 1084.32  951.36
 1117.72  951.96 1126.83     953 1178.45  955.39 1208.81  957.55 1220.96  961.79
#Mann= 3 , 0 , 0
       0     .09       0  923.07     .04       0  931.01     .09       0
Bank Sta=923.07,931.01
XS Rating Curve= 0 ,0
Exp/Cntr=0.3,0.1

Type RM Length L Ch R = 1 ,7315.2  ,3.71,91.44,11.6
XS GIS Cut Line= 6
     636935.4559    4335980.5286     636281.7439     4336421.033
     636170.6187    4336467.0926      636159.028    4336449.4835
      636108.706     4336464.976     635939.5623    4336735.3864
#Sta/Elev= 30
       0  962.47   55.29  959.21   79.87  956.56   95.23  953.11  110.59  952.46
   119.8  953.36  125.95  955.81  132.09  956.97  190.45  957.88  251.89  954.11
  322.54  951.44  334.83  950.31  405.48  951.15  439.27  950.16  460.78  948.63
  500.71  949.63  540.64  948.83  568.29  946.35  763.25  943.74  914.23  943.74
   924.9  943.74 1003.09  944.85 1030.69  948.62 1076.69  947.53 1088.96  949.81
 1101.23   950.8  1150.3  952.28 1239.24  956.62 1276.04  960.66 1306.71  961.97
#Mann= 3 , 0 , 0
       0     .09       0  914.23     .04       0   924.9     .09       0
Bank Sta=914.23,924.9
XS Rating Curve= 0 ,0
Exp/Cntr=0.3,0.1

Type RM Length L Ch R = 1 ,7223.76 ,12.85,91.44,210.53
XS GIS Cut Line= 6
     636925.4679    4335968.0932     636347.6903    4336354.7988
      636252.645    4336430.6883     636233.2888     4336401.963
     636101.0981    4336454.8115     635871.3658     4336721.628
#Sta/Elev= 30
       0  962.74   21.51  959.89   49.17   958.6   61.47  956.35   86.06  953.26
  107.57  952.78  126.01  956.75  187.48  957.65  331.93  950.89  396.47  951.48
  461.01  949.48  510.19  949.66  547.07  948.76  568.58  946.43  741.48  943.74
  830.94  943.74  840.74  943.74  958.87  944.48 1010.01  945.67 1028.38  947.59
 1046.75  946.96 1120.23  950.22 1236.57   953.3 1254.94   954.5 1270.25   954.2
 1288.62  955.89  1322.3  956.23 1328.42  957.76 1340.67  962.18 1349.85  963.49
#Mann= 3 , 0 , 0
       0     .09       0  830.94     .04       0  840.74     .09       0
Bank Sta=830.94,840.74
XS Rating Curve= 0 ,0
Exp/Cntr=0.3,0.1

Type RM Length L Ch R = 1 ,7132.32 ,131.89,91.44,327.95
XS GIS Cut Line= 6
     636919.1179    4335957.5098     636380.0452    4336340.3358
     635826.5487    4336505.5187      635231.602     4337101.835
     635037.1329    4337597.9298     634731.5385    4337951.1492
#Sta/Elev= 30
       0  962.45   21.43  958.99   79.59  953.32  107.14  953.18  131.62   957.1
  189.78  957.17  336.71   951.5  520.37  949.66  544.86  949.07  569.35  946.45
  746.08  943.74  759.04  943.74  975.53  946.25 1374.18  946.14 1543.63  947.82
 1580.25  946.68 1678.09  947.46 1699.49  949.38 1772.75  948.23 1796.75  950.17
 1972.72  949.06 2006.45  951.23 2052.44  949.39 2162.85  950.98 2285.61   950.5
  2404.3   953.1 2544.74  953.69 2684.26  957.98 3105.23  961.01 3151.32  963.39
#Mann= 3 , 0 , 0
       0     .09       0  746.08     .04       0  759.04     .09       0
Bank Sta=746.08,759.04
XS Rating Curve= 0 ,0
Exp/Cntr=0.3,0.1

Type RM Length L Ch R = 1 ,7040.88 ,65.75,91.44,21.91
XS GIS Cut Line= 6
     636998.8899    4335882.7649     636298.2076    4336220.6526
     636250.2049    4336258.7046     636212.7669    4336303.9219
     636068.7914    4336267.6603      635573.312    4336366.9533
#Sta/Elev= 30
       0  973.42    6.13  971.44    24.5  972.97   42.88  971.59   67.38  968.88
   82.69  964.33      98  964.81  150.07   956.8  199.07  954.37  235.82  957.21
  355.26  955.59  462.45  951.77  514.52  952.29  569.64  950.85  655.39  946.65
  868.51  944.01  875.41  944.02  903.92  943.53 1217.84  946.83 1248.46  948.98
 1291.34   956.8 1352.59  963.14 1370.97  970.04 1407.72  968.36 1426.09  969.58
 1444.47  968.28 1456.72  969.69 1484.28  968.41 1505.72  971.02 1551.66   972.2
#Mann= 3 , 0 , 0
       0     .09       0  868.51     .04       0  875.41     .09       0
Bank Sta=868.51,875.41
XS Rating Curve= 0 ,0
Exp/Cntr=0.3,0.1

Type RM Length L Ch R = 1 ,6949.44 ,115.21,91.44,37.31
XS GIS Cut Line= 6
     636883.0022    4335922.4524      636185.904    4336204.5932
      636178.794    4336209.4354      636096.461    4336252.1429
     636076.4352    4336246.9377      635793.975    4336293.9282
#Sta/Elev= 30
       0  964.55    9.21  962.26   18.42  959.15   27.63  957.32   79.81  954.91
   110.5  957.37  159.61  955.24  199.52  954.93  239.42   953.6   291.6  953.48
  377.55  950.95  429.73  951.45  506.47  947.96   534.1  947.33  546.37  946.45
  632.32  945.04  666.08  943.98  739.75  943.53  758.18  943.53  766.01  943.53
  823.25  943.54   877.2  945.59  919.85  945.49  971.64  946.57  992.96   946.2
 1056.93  947.91 1078.25  950.79 1102.62  956.81 1114.81   958.8  1160.5  963.09
#Mann= 3 , 0 , 0
       0     .09       0  758.18     .04       0  766.01     .09       0
Bank Sta=758.18,766.01
XS Rating Curve= 0 ,0
Exp/Cntr=0.3,0.1

Type RM Length L Ch R = 1 ,6858    ,20.64,91.44,128.04
XS GIS Cut Line= 6
     636851.2521    4335895.4649     636202.4846    4336070.5154
     636127.0782    4336131.6342     636128.6657    4336172.1156
     636077.8656    4336230.8532     635814.6125    4336262.1781
#Sta/Elev= 30
       0  964.32   21.48  960.17   33.75  959.62   52.16  957.94  168.76  953.58
  177.96  952.89  282.29  950.56  441.84  949.21  500.14  946.77  558.44  945.63
  638.22  944.87   693.2  946.43  726.57  945.13   738.7  943.78  800.75  943.85
  809.05  943.74  838.58  943.54  872.07  943.61  898.61  945.21  965.65  945.66
 1005.26  947.04 1063.16  948.24  1072.3  949.17 1075.35   950.1 1090.59  952.55
 1096.68  954.39 1111.92  956.84 1121.06  958.89 1139.34  961.16 1157.63  962.73
#Mann= 3 , 0 , 0
       0     .09       0  800.75     .04       0  809.05     .09       0
Bank Sta=800.75,809.05
XS Rating Curve= 0 ,0
Exp/Cntr=0.3,0.1

Type RM Length L Ch R = 1 ,6766.56 ,48.76,91.44,39.43
XS GIS Cut Line= 6
     636860.7771    4335868.4773     636184.7452    4336058.9863
     636146.3616    4336088.3753     636022.5014    4336139.5646
     636001.5209    4336133.4006       635809.85    4336190.7405
#Sta/Elev= 30
       0  962.82     9.2  961.72  116.55  955.07  177.89  953.62  226.96  951.56
   269.9  950.53  315.91  949.55  346.58   949.8  450.86  948.93  530.61  946.11
  644.09  944.75  702.36  945.43  741.64  944.82  765.93  945.69  793.35  945.73
  799.44  945.43  805.53   944.2  811.62  943.75  848.18  943.78  851.22  943.47
  857.02  943.78  884.73  943.78  906.59  945.43  988.44  947.82 1003.59  950.86
 1024.81  952.18 1049.06  952.91 1061.19  956.43  1091.5   961.1 1106.66  962.66
#Mann= 3 , 0 , 0
       0     .09       0  848.18     .04       0  857.02     .09       0
Bank Sta=848.18,857.02
XS Rating Curve= 0 ,0
Exp/Cntr=0.3,0.1

Type RM Length L Ch R = 1 ,6675.12 ,28.62,91.44,109.97
XS GIS Cut Line= 6
     636852.3435    4335850.5518     636160.8445    4336017.5404
     636030.8677    4336063.1811     636031.8761    4336088.2293
     636013.0083    4336111.4677     635801.4164    4336175.9899
#Sta/Elev= 30
       0  962.47  113.45  954.78  202.37  952.16   254.5  949.97  303.56  949.29
  337.29  949.95  364.89  947.66  417.01   947.9  438.48   947.4  453.81  948.68
  469.14  946.22  487.54  946.59   527.4  945.68  607.12  945.62  656.18  944.32
  696.05  944.47  720.46  945.29  741.65  944.71  793.12  945.32  860.93  943.35
   863.5  943.32  870.89  943.38  922.55  943.51  937.92   945.6 1008.58  947.77
 1023.94  950.94 1057.74  953.17 1070.03  955.92 1082.32  957.78  1128.4   963.3
#Mann= 3 , 0 , 0
       0     .09       0  860.93     .04       0  870.89     .09       0
Bank Sta=860.93,870.89
XS Rating Curve= 0 ,0
Exp/Cntr=0.3,0.1

Type RM Length L Ch R = 1 ,6583.68 ,25.35,91.44,71.8
XS GIS Cut Line= 6
      636850.756    4335833.0892      636149.452    4335999.0879
     635992.4876     4336053.526      635972.538     4336028.865
     635956.1073    4336017.4764     635776.0164    4336080.7397
#Sta/Elev= 30
       0  963.13   33.73  960.07  125.74  954.24     184  952.17  208.54  952.23
  266.81  949.45  297.47   949.3  331.21  950.49  364.94  947.22  456.94  946.58
  466.14  948.37  472.28  948.55  484.54  946.41  499.88   945.7  616.41  945.66
  741.83  944.03  826.41  944.84  894.93  943.57  905.74  943.21  908.33  943.55
  916.12  945.53  924.43  946.28  965.97  947.35 1011.42   950.2 1038.69  954.42
 1075.05  954.61 1081.11  956.29 1084.14  958.29  1090.2  959.71 1129.59  963.22
#Mann= 3 , 0 , 0
       0     .09       0  894.93     .04       0  908.33     .09       0
Bank Sta=894.93,908.33
XS Rating Curve= 0 ,0
Exp/Cntr=0.3,0.1

Type RM Length L Ch R = 1 ,6492.24 ,115.06,91.34,77.2
XS GIS Cut Line= 6
      636844.406    4335821.9767     636097.4328    4335987.7006
     636042.2302    4335982.6822     636021.8277    4335979.3025
     636011.7735    4335976.1275     635761.7288    4336061.6897
#Sta/Elev= 30
       0  963.26  113.69  954.64  190.52  951.53  224.32  951.52  261.19  949.19
   316.5  949.75   350.3  947.24   430.2  946.71  467.07  946.68  473.22  947.83
  482.44  948.14  494.73  946.27  503.95  945.75  614.57  945.66     633  944.82
  676.02  944.76  797.23  942.73  811.81  942.82  820.57  942.95  846.52  943.64
  879.45  945.53   953.2  947.75 1002.37  951.66 1026.95  954.56 1057.68  954.27
 1063.83  955.48 1069.97   958.7 1076.12   960.4  1100.7  962.64 1116.07  963.13
#Mann= 3 , 0 , 0
       0     .09       0  811.81     .04       0  820.57     .09       0
Bank Sta=811.81,820.57
XS Rating Curve= 0 ,0
Exp/Cntr=0.3,0.1

Type RM Length L Ch R = 1 ,6400.901,118.77,91.54,97.82
XS GIS Cut Line= 4
     636790.4309    4335629.8888     636046.9039    4335886.2266
     635850.8354    4335962.9395     635738.9746    4336043.0806
#Sta/Elev= 30
       0  962.89   73.73  957.82   187.4  952.67  245.77  951.72  270.35  952.08
  316.43  951.04   374.8  951.18  427.03  952.17  442.39  951.09  482.33   950.8
  534.56  949.07  546.84  948.34  556.06   946.9  565.28  948.59  571.42  948.66
  589.85  947.08  666.66  944.92  675.87  945.43  685.09  944.71  758.82  945.12
  807.83  942.81  810.77  942.71  820.04  942.75 1006.19  950.18 1027.59  952.86
 1067.34  954.39 1073.46  955.59 1085.69  959.42 1122.39   961.7 1134.62  963.12
#Mann= 3 , 0 , 0
       0     .09       0  807.83     .04       0  820.04     .09       0
Bank Sta=807.83,820.04
XS Rating Curve= 0 ,0
Exp/Cntr=0.3,0.1

Type RM Length L Ch R = 1 ,6309.36 ,63.54,91.44,79.43
XS GIS Cut Line= 5
     636609.4555    4335490.1004     636016.0271    4335770.9035
     636004.8637    4335796.8538     635859.2497    4335902.6991
     635675.4745    4336031.1744
#Sta/Elev= 30
       0  963.26   36.81  961.04  187.14  955.95  227.02   953.9  288.37  953.34
  408.02  949.01  444.83  948.92  500.05   947.6  509.26  946.83  515.39  948.08
  521.53  948.45  536.87  946.78  595.16   946.2  604.36  945.54  693.91   944.7
  718.32  942.71  728.22  942.71  736.91  942.71  757.99  944.14  785.45  943.98
  837.32  947.05  889.35  949.39  920.07  949.95  935.43  952.23  944.64  951.66
  950.79  951.96  996.86  957.63 1036.79  961.56 1052.15  961.24 1089.01  962.72
#Mann= 3 , 0 , 0
       0     .09       0  728.22     .04       0  736.91     .09       0
Bank Sta=728.22,736.91
XS Rating Curve= 0 ,0
Exp/Cntr=0.3,0.1

Type RM Length L Ch R = 1 ,6217.92 ,47.37,91.44,115.06
XS GIS Cut Line= 6
     636592.2576    4335474.2253     636114.4287    4335696.9905
     635955.7501    4335750.6031     635942.9024    4335779.2066
     635888.7156    4335794.6582     635594.7764    4336024.5598
#Sta/Elev= 30
       0  963.33    61.3  959.94  174.71  956.18  220.69  953.79   272.8  954.07
   343.3  950.88  505.75  946.72  521.07  948.64  542.43  946.29  630.74  944.97
   711.8  945.58  788.04  942.73  790.85  942.71  802.86  942.71  808.28   943.2
   817.1  946.01  914.78  949.36  926.99  951.43  942.25  950.64  975.83  952.82
 1006.35  956.65 1030.77  956.99 1046.03  958.13 1064.35  954.35 1082.66  954.24
 1088.77  955.91 1091.82  957.83 1110.14  959.54 1128.45  959.66 1158.97  962.53
#Mann= 3 , 0 , 0
       0     .09       0  788.04     .04       0  802.86     .09       0
Bank Sta=788.04,802.86
XS Rating Curve= 0 ,0
Exp/Cntr=0.3,0.1

Type RM Length L Ch R = 1 ,6126.48 ,86.59,91.44,92.42
XS GIS Cut Line= 6
     636569.7679    4335460.9961     636091.8006     4335684.446
     635951.5366    4335722.6032     635865.7063    4335720.2777
     635789.7131    4335731.4158     635608.0056    4335838.0281
#Sta/Elev= 30
       0  962.91   55.22  959.73  141.11  956.78  193.26   954.4   217.8  953.86
  260.74  954.03  411.05  948.39  500.01  946.33  506.15   946.3  512.28  947.04
  515.35  946.49  573.05  946.29  603.33  945.43  618.47  945.98  734.92  944.34
  743.54  943.67   751.8  942.83  756.99  943.58  805.67  946.39  836.39  946.47
  866.92  948.08  882.19  949.88   894.4  950.48  915.77  950.32  973.78  951.64
  995.16  954.77 1007.37     955 1019.58  956.08 1044.01  960.13 1047.06  961.52
#Mann= 3 , 0 , 0
       0     .09       0  743.54     .04       0  756.99     .09       0
Bank Sta=743.54,756.99
XS Rating Curve= 0 ,0
Exp/Cntr=0.3,0.1

Type RM Length L Ch R = 1 ,6035.04 ,42.75,42.03,42.67
XS GIS Cut Line= 6
      636536.695    4335434.5378     636063.0989    4335639.0048
     635892.7549     4335636.371     635870.8959    4335630.9543
     635848.4371    4335632.4022     635622.5577    4335787.7572
#Sta/Elev= 30
       0  963.19  101.33  957.75  162.74  956.62  205.73  954.37  334.69  950.23
  374.61  950.35  442.16   948.8     479  950.98  494.36  950.44  503.57  948.26
  512.78  947.92  570.61  951.32  597.99  948.03  610.16  945.18  622.33  945.77
  689.19  943.27  698.11  942.75  703.47  943.42   725.7  944.66   795.3  945.06
  831.85  946.59  850.13  946.09  871.45  949.66  886.68   950.1  904.96  952.51
  932.37  953.09  956.74  955.57  984.15  958.64  990.25   960.7 1005.48  962.68
#Mann= 3 , 0 , 0
       0     .09       0  689.19     .04       0  703.47     .09       0
Bank Sta=689.19,703.47
XS Rating Curve= 0 ,0
Exp/Cntr=0.3,0.1

Type RM Length L Ch R = 1 ,5993.011,18.5,17.28,18.1
XS GIS Cut Line= 6
     636482.4553    4335405.4335     636047.1266    4335604.8411
     635928.6859    4335594.0669     635910.5884    4335605.6557
     635861.0583     4335588.934      635617.266    4335752.0384
#Sta/Elev= 30
       0  962.81    70.6  958.03  153.47  955.34  211.79  955.26  270.11  953.32
  285.45  951.27  297.73  952.99  316.15  953.22   340.7  952.65  349.91   950.3
  365.26  951.62  414.37  951.71  481.88  947.99  564.21  948.95  585.56  945.13
  606.97  943.92  636.49  944.33  643.76  943.06   648.3  942.46   654.1  942.96
  700.95  944.71  801.78  945.41  835.39  949.51  853.72  949.89  862.89  951.98
  875.11  951.78  890.39  953.69  933.16  954.42  945.38  958.11  969.83  962.26
#Mann= 3 , 0 , 0
       0     .09       0  643.76     .04       0   654.1     .09       0
Bank Sta=643.76,654.1
XS Rating Curve= 0 ,0
Exp/Cntr=0.3,0.1

Type RM Length L Ch R = 1 ,5975.728,66.06,32.13,8.62
XS GIS Cut Line= 6
     636438.7989    4335357.8084     636040.6279    4335576.6795
     635928.3067      4335575.76     635911.1087    4335585.0204
     635866.1295     4335567.161     635606.6827    4335738.8092
#Sta/Elev= 30
       0  963.24   52.19  959.72   95.17  959.37  138.15  956.37  205.69  955.55
  211.83  956.09  230.25  960.39  251.74  960.64   276.3  959.01  328.49  951.22
  349.98  953.36  386.82  953.82  426.73  952.17  454.36  947.71   499.9  948.05
  530.26  945.82  572.27  944.85  597.97   942.5   608.2  942.17  612.88  942.57
  617.55  943.91  622.39   943.3  643.75  944.31  782.52  945.68   803.8  949.41
  828.11  949.72  840.26  952.82   913.2  955.14  931.43  960.47  949.67     963
#Mann= 3 , 0 , 0
       0     .09       0  597.97     .04       0  612.88     .09       0
Bank Sta=597.97,612.88
XS Rating Curve= 0 ,0
Exp/Cntr=0.3,0.1

Type RM Length L Ch R = 1 ,5943.6  ,77.73,91.44,96.98
XS GIS Cut Line= 6
     636177.6547    4335384.2668     635868.4389    4335548.5402
     635864.7679     4335555.615     635858.0283    4335562.8387
     635831.5255    4335588.0101     635605.3598    4335728.2258
#Sta/Elev= 30
       0  963.21   33.79  955.81   58.36  959.39  175.07  957.16   193.5  954.65
  199.64  953.08  205.79  950.53  239.57  947.18  248.79  945.27     258  947.34
  285.64  949.88     301   952.5  307.14   952.4   322.5   950.5  334.79  944.56
  340.93     943  347.07   942.4  350.14  941.98  355.46  942.48  367.99  944.08
  389.31  944.96  502.42  946.25  514.66   947.8  520.77  949.33  551.36  950.11
  563.59  952.99  633.94  955.23  640.06  956.38   652.3  960.11  670.65   962.5
#Mann= 3 , 0 , 0
       0     .09       0  347.07     .04       0  355.46     .09       0
Bank Sta=347.07,355.46
XS Rating Curve= 0 ,0
Exp/Cntr=0.3,0.1

Type RM Length L Ch R = 1 ,5852.16 ,96.57,91.44,70.28
XS GIS Cut Line= 5
     636183.1117    4335343.5209     635867.9228    4335464.2439
     635833.6287    4335471.1028     635801.7711    4335482.2068
     635570.3355    4335680.0716
#Sta/Elev= 30
       0  963.05   30.68  959.14  113.53  959.49  153.42  957.48  202.51     956
  211.72  954.81  220.92  950.89   242.4  947.77  254.67  948.61  266.95   947.3
  276.15  947.22  285.36  948.79  303.77  950.12  325.24  950.65  331.38  948.99
  344.38  942.74  346.26   941.9  356.79  942.59  400.09  944.06  488.44  945.78
  509.75  947.61  561.52  948.72  588.92  950.11  598.05  951.05  607.19  953.16
  649.82  955.39  665.04  956.76  674.18  958.34  692.45  959.52  710.71  963.35
#Mann= 3 , 0 , 0
       0     .09       0  344.38     .04       0  356.79     .09       0
Bank Sta=344.38,356.79
XS Rating Curve= 0 ,0
Exp/Cntr=0.3,0.1

Type RM Length L Ch R = 1 ,5760.72 ,91.16,91.44,85.36
XS GIS Cut Line= 5
      636057.699    4335205.4081     635818.5539    4335384.6482
     635805.9664    4335391.3916     635798.3933    4335397.2224
      635565.573    4335661.0215
#Sta/Elev= 30
       0  963.32     6.1  960.56    12.2   959.1   42.69  957.38   70.14   957.1
   76.24  957.64   91.49  960.45  109.79  959.85  158.58  954.94  189.07  949.16
  225.67  946.76  256.17  946.81  277.51  946.27  289.71  944.88  304.57  942.26
  307.43  941.88  315.53   942.2  365.53  943.98  426.72  944.06  445.08  946.39
  478.73  946.63  494.03   947.9  521.57  948.13  539.92  948.91  570.52  952.76
  598.06  954.18  616.41   955.7  647.01  957.01  665.36  959.59  674.54  962.28
#Mann= 3 , 0 , 0
       0     .09       0  304.57     .04       0  315.53     .09       0
Bank Sta=304.57,315.53
XS Rating Curve= 0 ,0
Exp/Cntr=0.3,0.1

Type RM Length L Ch R = 1 ,5669.28 ,94.27,91.44,37.78
XS GIS Cut Line= 6
     635903.7111    4335162.5455     635746.0131    4335334.3715
     635733.5635    4335345.3829     635724.6978    4335351.5764
     635645.4666    4335445.8098     635495.7228     4335662.609
#Sta/Elev= 30
       0  963.14   27.62  959.11   33.76  957.74   42.96  954.52   55.24  952.53
   67.51   951.3   79.79  948.53  101.27  948.28  116.61  950.38  122.75  950.34
   147.3  947.95  174.92  947.09  187.19  945.48  208.67   945.2  241.53  943.11
   244.3  942.43  249.84   941.6  255.25  942.17  350.74  942.74  368.76  945.23
  408.28  946.46  432.79  947.87  484.88  952.21  515.52  951.84  546.16  956.02
  570.67  958.09  585.98  958.81  641.13  959.84   644.2  960.42  647.26  961.78
#Mann= 3 , 0 , 0
       0     .09       0   244.3     .04       0  255.25     .09       0
Bank Sta=244.3,255.25
XS Rating Curve= 0 ,0
Exp/Cntr=0.3,0.1

Type RM Length L Ch R = 1 ,5577.84 ,127.15,91.44,46.01
XS GIS Cut Line= 6
     635810.0485    4335029.1953     635674.5273    4335274.7558
     635661.2946    4335289.2754     635686.4103    4335338.2348
      635670.866    4335357.0864     635475.0853     4335659.434
#Sta/Elev= 30
       0  962.93   42.68  956.82   57.92  955.25   76.22  953.94   91.46  953.74
  134.14  955.32  152.43  955.45  158.53  954.99  182.92  950.19  189.02   949.3
  210.36  949.83   213.4  949.31   219.5  947.29  222.55  946.76  271.33   943.4
  286.09  941.96  288.89  941.61  294.51   941.8  339.86  942.29  425.37  941.82
  449.79  943.78   468.1  944.04  483.37  946.04  501.68  947.57  535.26  947.77
  596.31   951.4  623.78  954.19   648.2  958.27  718.41  959.33  739.78  961.13
#Mann= 3 , 0 , 0
       0     .09       0  286.09     .04       0  294.51     .09       0
Bank Sta=286.09,294.51
XS Rating Curve= 0 ,0
Exp/Cntr=0.3,0.1

Type RM Length L Ch R = 1 ,5486.4  ,31.83,91.44,102.23
XS GIS Cut Line= 6
     635775.1234    4334967.2827     635577.3246    4335238.3874
     635579.7059    4335296.8605     635623.0976    4335296.5959
     635651.9373    4335333.6376     635459.2103     4335659.434
#Sta/Elev= 30
       0  962.94   97.63  957.92  115.93  957.38  149.49   959.8  164.75  959.36
  195.25  956.12  219.66  951.55  228.81  951.16  247.12   946.5  250.17  946.07
  394.11  941.73  416.85   941.7  422.92   941.6  425.89  941.65  485.99  942.14
   556.2   941.7  571.46  943.96  595.88  944.62  605.04  946.35  611.15  946.99
   672.2  948.48  711.89  950.78  748.52  955.15  769.89  958.19  785.15  958.07
  830.94  959.16   840.1  959.83  858.42  960.24  861.47  960.47  864.52  961.42
#Mann= 3 , 0 , 0
       0     .09       0  416.85     .04       0  425.89     .09       0
Bank Sta=416.85,425.89
XS Rating Curve= 0 ,0
Exp/Cntr=0.3,0.1

Type RM Length L Ch R = 1 ,5394.96 ,41.29,91.44,95.06
XS GIS Cut Line= 6
     635773.5359    4334951.4076     635569.2394    4335230.5999
     635573.8079    4335285.9684     635567.1933    4335291.7893
     635583.5975    4335345.4998     635422.6977    4335614.9839
#Sta/Elev= 30
       0  962.79   18.37  962.72   67.35  960.22  125.52  957.95  162.26  960.13
  168.39  960.32  177.57  959.95  195.94  956.89  214.31  955.31  220.43  954.17
  229.62  951.63   238.8  950.95  244.92  949.73  247.99  949.52  263.29  946.16
  266.36  945.92  422.15  941.52   469.5  941.73   480.5  941.77  487.96   943.6
  493.84  944.19  523.91  945.12   557.7  947.29  594.56     948  649.85   950.9
  683.64  954.14     699  954.72  714.36  956.05  726.65  956.64  781.94  962.92
#Mann= 3 , 0 , 0
       0     .09       0   469.5     .04       0   480.5     .09       0
Bank Sta=469.5,480.5
XS Rating Curve= 0 ,0
Exp/Cntr=0.3,0.1

Type RM Length L Ch R = 1 ,5303.52 ,96.09,91.44,78.49
XS GIS Cut Line= 4
      635761.365    4334946.6451     635535.5511    4335269.4648
       635506.98    4335297.5196     635287.7599    4335552.5422
#Sta/Elev= 30
       0  962.76   24.43  962.45   42.76  961.25   91.62  959.28     113  957.95
  122.16     958  171.02  960.87  195.45  957.07  213.78  955.07  225.99  951.77
  235.15  951.11  250.42  947.93  262.64  946.09  332.88  943.78  402.54  942.24
  408.26  941.55  413.98  942.25   419.7  943.25  428.28  943.63  482.92   944.8
   519.6  946.03  559.35  946.22   663.3  950.37  696.92  953.05  712.21   954.7
   727.5  954.81  739.73  957.57  745.84  959.52  755.01  961.64   770.3  963.06
#Mann= 3 , 0 , 0
       0     .09       0  402.54     .04       0  413.98     .09       0
Bank Sta=402.54,413.98
XS Rating Curve= 0 ,0
Exp/Cntr=0.3,0.1

Type RM Length L Ch R = 1 ,5212.08 ,75.93,91.44,112.2
XS GIS Cut Line= 4
     635678.6826    4334936.9437     635461.2377    4335207.2875
      635418.577    4335295.7891     635239.6497    4335523.8789
#Sta/Elev= 30
       0  963.39   24.56  959.64   42.98  959.29   67.55  958.17  132.02  957.62
  153.51  954.97  162.72  952.71  165.79  952.28  175.01  952.01  211.85  948.84
  254.83  946.04  285.54  944.55  359.22  942.33  365.36  941.66  368.43  942.11
  374.57  942.94  380.71   943.3  411.42  944.27   475.7  944.41  487.91  945.88
  509.27  945.21  521.48  945.34  613.02   949.4  637.43  950.89  674.05  954.13
  689.31  956.08  707.62  959.51  716.77  960.24  722.88  961.13  735.08  963.38
#Mann= 3 , 0 , 0
       0     .09       0  359.22     .04       0  368.43     .09       0
Bank Sta=359.22,368.43
XS Rating Curve= 0 ,0
Exp/Cntr=0.3,0.1
